--- PTLCKFK.prj (project) ---

Proj Title=PTLCKFK
Current Plan=p01
Default Exp/Contr=0,0
English Units
Geom File=g01
Flow File=f01
Plan File=p01
BEGIN DESCRIPTION:
END DESCRIPTION:
DSS Export Rating Curves= 0
DSS Export Rating Curve Sorted= 0
DSS Export Volume Flow Curves= 0
DXF OffsetX= 0
DXF OffsetY= 0
DXF ScaleX= 0
DXF ScaleY= 0

--- PTLCKFK.p01 (plan) ---

Plan Title=Floodplain
Program Version=4.00
Geom File=g01
Flow File=f01
K Sum by GR=0
Std Step Tol=0.01
Critical Tol=0.01
Num of Std Step Trials=20
Max Error Tol=0.3
Flow Tol Ratio=0.001
Split Flow NTrial=30
Split Flow Tol=0.02
Split Flow Ratio=0.02
Log Output Level=0
Friction Slope Method=1
Unsteady Friction Slope Method=2
Unsteady Bridges Friction Slope Method=1
Global Log Level=0
CheckData=False
Run HTab=0
Run UNet=0
Run PostProcess=0
UNET Theta=0
UNET Theta Warmup=0
UNET ZTol=0
UNET ZSATol=0
UNET MxIter=0
UNET MaxInSteps=0
UNET DtIC=0
UNET DtMin=0
UNET MaxCRTS=0
UNET WFStab=0
UNET SFStab=0
UNET WFX=0
UNET SFX=0
UNET DSS MLevel=0
UNET DZMax Abort=0
UNET Convert EG Bridges=0
UNET Use Existing IB Tables=0
UNET Froude Limit=0
UNET Froude Power=0
Write IC File=0
Echo Input=False
Echo Output=False
Write Detailed=0

--- PTLCKFK.f01 (steady flow) ---

Flow Title=NFF Regression Equation
Program Version=4.10
Number of Profiles= 1
Profile Names=P100yr
River Rch & RM=PTLCKFK,Main            ,10362.3
865.4843
River Rch & RM=PTLCKFK,Main            ,8255.2
959.3076
River Rch & RM=PTLCKFK,Main            ,6638.4
1057.031
River Rch & RM=PTLCKFK,Main            ,5641.7
1143.386
River Rch & RM=PTLCKFK,Main            ,4248.3
1223.218
Boundary for River Rch & Prof#=PTLCKFK,Main            , 1
Up Type= 0
Dn Type= 3
Dn Slope=0.011
DSS Import GetInterval= 0
DSS Import GetPeak= 0
DSS Import FillOption= 0

--- PTLCKFK.g01 (geometry) ---

Geom Title=USGS 10m DEM
Program Version=4.10

River Reach=PTLCKFK         ,Main
Reach XY= 30
     1830957.333      478369.347     1830624.868      478640.181
     1830483.375      478675.771     1830244.731      479211.037
     1830028.104      479336.771     1829919.606      479636.759
     1829787.557      479829.395     1829648.306      479963.965
     1829410.458      480061.188     1829326.257      480174.035
     1829190.578      480205.035     1828872.264       480475.25
     1828729.503      480690.203      1828718.33      480957.814
     1828654.789      481097.397     1828225.969        481440.8
     1827636.066      481616.483     1827105.898      481638.302
     1826852.078      481695.586     1826824.134      481756.596
     1826586.587      481835.233     1826285.513      481850.818
      1826048.24      481949.875     1825747.637      482000.876
     1825416.039      482140.199     1825320.553      482237.855
     1824826.196      482286.032     1823700.602       482538.55
     1822855.338      482419.806     1822578.146      482598.808

Type RM Length L Ch R = 1 ,10362.3 ,164.8,173.8,182.6
XS GIS Cut Line= 2
     1830867.961      478301.157     1831024.546      478441.662
#Sta/Elev= 25
       0  781.95     9.6  781.47    19.1  781.24    28.7  781.31    38.2  780.85
    47.8  778.28    57.4  776.92    66.9  776.83    76.5   776.9    86.1  777.06
    95.6  776.89   105.2  775.81   105.7  775.76   114.8  774.82   120.7  775.11
   124.3  775.29   133.9  777.45   143.4  781.06     153  786.02   162.6  791.62
   172.1  797.44   181.7  804.16   191.3   811.4   200.8  817.97   210.4  823.15
#Mann= 3 , 0 , 0
       0      .1       0   105.7    .045       0   120.7      .1       0
Bank Sta=105.7,120.7
XS Rating Curve= 0 ,0
Exp/Cntr=0.3,0.1

Type RM Length L Ch R = 1 ,10188.5 ,25.6,36.9,47.2
XS GIS Cut Line= 3
     1830773.909      478392.972     1830797.525      478439.048
     1830844.921      478538.007
#Sta/Elev= 21
       0  777.97     8.6  777.88    17.3  777.49    25.9  776.88    34.5  776.47
    43.2  776.22    51.8  775.97    60.9  775.86    70.1  775.56    79.2  774.58
    87.9  772.93    88.4  772.84    97.5  773.07   102.9  774.96   106.6  776.26
   115.8  781.38   124.9  786.95   134.1  792.46   143.2  798.24   152.4  804.01
   161.5  809.99
#Mann= 3 , 0 , 0
       0      .1       0    87.9    .045       0    97.5      .1       0
#XS Ineff= 2 , 0
           48.82  780.33
Permanent Ineff=
       F       F
Bank Sta=87.9,97.5
XS Rating Curve= 0 ,0
Exp/Cntr=0.3,0.1

Type RM Length L Ch R = 1 ,10151.6 ,29.3,29.2,29.3
XS GIS Cut Line= 3
     1830763.262      478396.524     1830783.721      478438.759
     1830784.095      478568.399
#Sta/Elev= 21
       0  777.91     9.4     778    18.8  777.94    28.2  777.69    37.5  777.32
    46.9  776.93    56.2  776.82    65.4  776.54    74.7  775.76      84  774.06
    93.2  772.08    96.6  771.81   102.5  771.33   111.6  772.91     121  774.75
   130.3  775.66   139.5  776.33   148.8  778.94     158  783.96   167.3  790.07
   176.6  796.21
#Mann= 3 , 0 , 0
       0      .1       0    93.2    .045       0   111.6      .1       0
Bank Sta=93.2,111.6
XS Rating Curve= 0 ,0
Exp/Cntr=0.3,0.1

Type RM Length L Ch R = 1 ,10122.4 ,95.2,78.3,62.1
XS GIS Cut Line= 3
     1830737.097      478402.338     1830757.556      478444.574
     1830757.931      478574.213
#Sta/Elev= 22
       0  778.55     9.4   778.5    18.8  778.13    28.2  777.67    37.5  777.42
    46.9   777.4    56.2  777.21    65.4  776.85    74.7  776.22      84   774.8
    93.2  772.63   102.5  770.94   103.8  770.88   111.8  770.49   118.8  771.35
     121  771.62   130.3  773.63   139.5  775.19   148.8   775.8     158  776.23
   167.3  777.58   176.6  780.87
#Mann= 3 , 0 , 0
       0      .1       0   102.5    .045       0   118.8      .1       0
Bank Sta=102.5,118.8
XS Rating Curve= 0 ,0
Exp/Cntr=0.3,0.1

Type RM Length L Ch R = 1 ,10044.1 ,102.8,108,113
XS GIS Cut Line= 2
     1830620.963      478467.173     1830742.317      478610.923
#Sta/Elev= 23
       0  775.39     9.4  774.84    18.8  774.31    28.2  773.71    37.6  773.08
      47  772.44    56.4  772.24    65.8  772.53    75.2  773.05    84.7  773.26
    94.1     772   103.5  769.82   105.2  769.68   112.9  769.07   120.2  769.73
   122.3  769.92   131.7  772.09   141.1  774.01   150.5  775.19   159.9  775.46
   169.3  776.95   178.7  782.34   188.1  791.07
#Mann= 3 , 0 , 0
       0     .07       0   103.5    .045       0   122.3      .1       0
#XS Ineff= 2 , 0
            84.7  775.25
Permanent Ineff=
       F       F
Bank Sta=103.5,122.3
XS Rating Curve= 0 ,0
Exp/Cntr=0.3,0.1

Type RM Length L Ch R = 1 ,9936.1  ,132.9,125.2,117.1
XS GIS Cut Line= 4
     1830540.754      478510.923     1830617.317      478616.132
     1830643.879      478667.694     1830670.963      478697.382
#Sta/Elev= 28
       0  775.63     9.3  775.01    18.6   774.4    27.9  773.78    37.2  773.08
    46.5  772.41    55.8  771.82    65.1  771.27    74.4  770.83    83.6  770.46
    92.9  770.08   102.2  769.85   111.5  770.31   120.8  771.06   130.1  771.35
   139.8  770.33   146.7  768.91   149.4  768.35   159.1  767.12   161.7  767.33
   168.8   767.9   178.4  770.87   188.1  772.56   196.2  773.67   204.2  776.46
   212.2   781.7   220.3  788.45   228.3  794.79
#Mann= 3 , 0 , 0
       0     .08       0   149.4    .045       0   168.8      .1       0
Bank Sta=149.4,168.8
XS Rating Curve= 0 ,0
Exp/Cntr=0.3,0.1

Type RM Length L Ch R = 1 ,9811    ,99.2,94.4,89.9
XS GIS Cut Line= 2
     1830430.338      478576.028     1830609.504      478744.778
#Sta/Elev= 29
       0  784.53     9.5  781.65    18.9  778.51    28.4  776.05    37.9  775.27
    47.3  775.14    56.8  774.98    66.3  774.51    75.7  773.73    85.2  771.51
    94.7  766.97   102.7  765.18   104.1  764.87   113.6  764.66   117.7  765.17
   123.1  765.84   132.5  768.54     142  770.33   151.5  770.41   160.9  770.48
   170.4  770.54   179.9  770.62   189.3  770.61   198.8  770.58   208.3  770.42
   217.7  771.28   227.2  774.95   236.7  780.52   246.1  786.37
#Mann= 3 , 0 , 0
       0      .1       0   102.7    .045       0   117.7      .1       0
Bank Sta=102.7,117.7
XS Rating Curve= 0 ,0
Exp/Cntr=0.3,0.1

Type RM Length L Ch R = 1 ,9716.5  ,75.2,72.5,69.9
XS GIS Cut Line= 2
     1830376.277      478678.843     1830555.223      478787.047
#Sta/Elev= 25
       0  776.64     9.5  773.84      19  772.72    28.5  772.85      38  773.03
    47.5  773.02      57  772.85    66.5  772.13      76  767.85    81.1  765.74
    85.6  763.87      95   762.9    96.1     763   104.6  763.77   114.1   765.7
   123.6  766.98   133.1  767.24   142.6  767.51   152.1  767.82   161.6  768.18
   171.1   768.5   180.6  768.45   190.1  768.36   199.6  770.35   209.1  774.72
#Mann= 3 , 0 , 0
       0     .08       0    85.6    .045       0   104.6     .06       0
Bank Sta=85.6,104.6
XS Rating Curve= 0 ,0
Exp/Cntr=0.3,0.1

Type RM Length L Ch R = 1 ,9644    ,22.3,22.3,22.4
XS GIS Cut Line= 2
     1830342.513      478753.925     1830524.175      478836.607
#Sta/Elev= 24
       0  772.92     9.5  772.67      19  773.08    28.5  773.64      38  773.85
    47.5  773.13      57   771.1    66.5  765.61    71.5   763.9      76  762.37
    85.5  761.86    86.5  761.95      95  762.71   104.6  764.28     114  765.25
   123.6  765.53   133.1  765.86   142.6  766.34   152.1  766.81   161.6  767.29
   171.1  767.19   180.6   767.3   190.1  770.04   199.6  775.38
#Mann= 3 , 0 , 0
       0     .06       0      76    .045       0      95     .06       0
Bank Sta=76,95
XS Rating Curve= 0 ,0
Exp/Cntr=0.3,0.1

Type RM Length L Ch R = 1 ,9621.7  ,18.9,18.6,18.3
XS GIS Cut Line= 2
      1830334.96      478774.993     1830516.622      478857.675
#Sta/Elev= 24
       0     773     9.5  772.52      19  772.82    28.5  773.23      38   773.3
    47.5   772.6      57  769.53    66.5  764.21    69.6  763.38      76  761.66
    84.6  761.61    85.5   761.6      95  762.68   104.6  764.21     114  764.78
   123.6  765.02   133.1  765.45   142.6  766.03   152.1  766.66   161.6  766.92
   171.1  766.78   180.6  768.14   190.1  772.78   199.6  778.99
#Mann= 3 , 0 , 0
       0     .06       0    69.6    .045       0      95     .06       0
Bank Sta=69.6,95
XS Rating Curve= 0 ,0
Exp/Cntr=0.3,0.1

Type RM Length L Ch R = 1 ,9603    ,17.8,17.1,16.3
XS GIS Cut Line= 3
     1830309.269       478785.76     1830336.579      478797.222
     1830497.144      478867.612
#Sta/Elev= 25
       0  781.51     7.4  777.07    14.8  774.45    22.2  773.17    29.6  772.42
    39.4   771.7    49.1  770.94    58.8  770.62    68.6  769.57    78.3  766.26
    88.1  762.63    88.9  762.54    97.8  761.55   103.9  761.71   107.5   761.8
   117.3  763.06     127  764.33   136.8  764.55   146.5   764.6   156.2  765.02
     166  765.75   175.7  766.32   185.5  766.53   195.2  767.62   204.9  771.85
#Mann= 3 , 0 , 0
       0     .06       0    88.9    .045       0   107.5     .06       0
Bank Sta=88.9,107.5
XS Rating Curve= 0 ,0
Exp/Cntr=0.3,0.1

Type RM Length L Ch R = 1 ,9586    ,36.9,36.9,36.9
XS GIS Cut Line= 3
     1830297.595      478802.421     1830473.033      478872.444
     1830487.394      478877.426
#Sta/Elev= 25
       0  782.61     9.4  777.76    18.9  773.45    28.3  769.48    37.8  767.29
    47.2  766.24    56.7  765.73    66.1  765.16    75.6  764.71      85  763.63
      93  762.19    94.4  761.94   103.9  761.48     108  761.92   113.3  762.49
   122.8  763.68   132.2  764.19   141.7  764.23   151.1  764.32   160.6  764.77
     170  765.43   179.4  766.08   188.9  766.44   196.5  767.33   204.1  770.67
#Mann= 3 , 0 , 0
       0     .06       0    94.4    .045       0     108     .06       0
Bank Sta=94.4,108
XS Rating Curve= 0 ,0
Exp/Cntr=0.3,0.1

Type RM Length L Ch R = 1 ,9549    ,65.9,65.8,65.7
XS GIS Cut Line= 2
     1830281.297      478835.414     1830464.549      478908.556
#Sta/Elev= 24
       0  777.65     9.4   773.8    18.8  769.78    28.2  766.68    37.6  765.21
      47  764.82    56.4  764.34    65.8  764.02    75.2  763.63    84.6  762.35
    91.7  761.18      94   760.8   103.4  760.12   106.7  760.19   112.8  760.33
   122.1  761.69   131.5  763.26   140.9  763.96   150.3  764.33   159.7  764.47
   169.1  764.81   178.5  765.49   187.9   766.3   197.3  768.88
#Mann= 3 , 0 , 0
       0     .06       0      94    .045       0   112.8     .06       0
Bank Sta=94,112.8
XS Rating Curve= 0 ,0
Exp/Cntr=0.3,0.1

Type RM Length L Ch R = 1 ,9483.3  ,57.6,58.4,59
XS GIS Cut Line= 2
     1830249.894      478894.093      1830435.31       478967.01
#Sta/Elev= 24
       0  771.83     9.5   768.9      19  766.66    28.5  765.59      38  765.07
    47.4  764.55    56.9  764.03    66.4  763.51    75.9  763.03    85.4  762.16
    94.9  760.76   100.6   760.2   104.4  759.83   113.8  759.86   115.6  759.97
   123.3  760.43   132.8   762.4   142.3  763.22   151.8  763.57   161.3  763.86
   170.8  764.47   180.3  765.11   189.8  765.64   199.2  767.69
#Mann= 3 , 0 , 0
       0     .08       0   100.6    .045       0   115.6      .1       0
Bank Sta=100.6,115.6
XS Rating Curve= 0 ,0
Exp/Cntr=0.3,0.1

Type RM Length L Ch R = 1 ,9424.9  ,21.3,21.4,21.3
XS GIS Cut Line= 2
     1830263.409      478959.437     1830395.432      479016.269
#Sta/Elev= 18
       0  765.65     9.6  764.79    19.2  763.86    28.8  763.05    38.3   762.6
    47.9  762.31    57.5  761.59      65  760.62    67.1  760.35    76.7  759.72
      80  760.04    86.2  760.65    95.8  761.96   105.4  762.46     115  762.56
   124.6  762.89   134.2  763.54   143.7  764.02
#Mann= 3 , 0 , 0
       0     .08       0      65    .045       0    86.2      .1       0
Bank Sta=65,86.2
XS Rating Curve= 0 ,0
Exp/Cntr=0.3,0.1

Type RM Length L Ch R = 1 ,9403.5  ,12.5,9.8,7.1
XS GIS Cut Line= 2
     1830251.086      478977.325     1830383.109      479034.157
#Sta/Elev= 17
       0  765.54     9.6  764.56    19.2  763.53    28.8  762.78    38.3  762.25
    47.9  761.98    57.5  761.71    67.1  760.57    71.2   759.9    76.7     759
    86.2  758.73    95.8  760.06   105.4  761.66     115  762.33   124.6  762.68
   134.2  763.13   143.7  763.41
#Mann= 3 , 0 , 0
       0     .06       0    71.2    .045       0    95.8     .06       0
Bank Sta=71.2,95.8
XS Rating Curve= 0 ,0
Exp/Cntr=0.3,0.1

Type RM Length L Ch R = 1 ,9393.7  ,16,16,16
XS GIS Cut Line= 3
     1830240.989      478994.419     1830361.408      479029.873
      1830398.96      479046.889
#Sta/Elev= 21
       0     765     9.7  764.43    19.3  763.63      29  762.95    38.6  762.36
    48.3  761.92    57.9   761.5    67.6  760.73      75  759.54    77.2  759.18
    86.9  758.17      90  758.45    96.6  759.04   106.2  761.13   115.9  762.06
   125.5  762.51   133.8   762.9     142  763.25   150.3  763.38   158.5  763.96
   166.8  767.34
#Mann= 3 , 0 , 0
       0      .1       0    77.2    .045       0    96.6     .06       0
Bank Sta=77.2,96.6
XS Rating Curve= 0 ,0
Exp/Cntr=0.3,0.1

Type RM Length L Ch R = 1 ,9377.7  ,36.9,36.5,36.1
XS GIS Cut Line= 2
     1830235.822      479009.524     1830395.159      479056.436
#Sta/Elev= 20
       0  764.42     9.8  764.36    19.5  763.76    29.3  763.15    39.1  762.56
    48.8  762.04    58.6  761.44    68.4  760.46    75.9  759.22    78.2  758.84
    87.9  758.02    90.9  758.28    97.7  758.86   107.5  760.62   117.2  761.85
     127   762.4   136.8  762.88   146.6  763.17   156.3  763.78   166.1  767.25
#Mann= 3 , 0 , 0
       0      .1       0    78.2    .045       0    97.7     .06       0
Bank Sta=78.2,97.7
XS Rating Curve= 0 ,0
Exp/Cntr=0.3,0.1

Type RM Length L Ch R = 1 ,9341.2  ,33,35.2,37.3
XS GIS Cut Line= 2
     1830227.434      479046.598     1830395.797      479092.983
#Sta/Elev= 21
       0  763.51     9.7  762.94    19.4  762.76    29.1  762.23    38.8  761.71
    48.5  761.11    58.2  760.57    67.9  759.43    75.6  758.18    77.6  757.85
    87.3  757.24    90.6   757.6      97  758.29   106.7  760.24   116.4  761.54
   126.1   762.2   135.8   762.6   145.5  762.98   155.2  765.05   164.9  769.96
   174.6  776.22
#Mann= 3 , 0 , 0
       0     .08       0    77.6    .045       0    90.6     .06       0
Bank Sta=77.6,90.6
XS Rating Curve= 0 ,0
Exp/Cntr=0.3,0.1

Type RM Length L Ch R = 1 ,9306    ,26.8,26.7,26.8
XS GIS Cut Line= 2
     1830195.656      479063.053     1830379.823      479133.595
#Sta/Elev= 24
       0  764.96     9.4  763.71    18.8  762.95    28.2  762.16    37.6  761.42
      47  760.97    56.4  760.72    65.7  760.37    75.1  760.18    84.5  759.93
    93.9   758.8   100.4  757.71   103.3  757.22   112.7  757.08   115.4  757.59
   122.1  758.86   131.5  760.81   140.9  761.96   150.3   762.3   159.6  762.44
     169  762.59   178.4  764.98   187.8  769.56   197.2  774.66
#Mann= 3 , 0 , 0
       0      .1       0   100.4    .045       0   115.4     .08       0
Bank Sta=100.4,115.4
XS Rating Curve= 0 ,0
Exp/Cntr=0.3,0.1

Type RM Length L Ch R = 1 ,9279.2  ,39.8,39.1,37.8
XS GIS Cut Line= 2
     1830181.453      479085.778      1830365.62       479156.32
#Sta/Elev= 24
       0  771.57     9.4  766.42    18.8  762.17    28.2   759.9    37.6  759.35
      47  759.22    56.4  759.26    65.7  759.13    75.1  759.08    84.5  758.98
    93.9  758.27   100.9  757.28   103.3  756.94   112.7   756.4   115.9  756.95
   122.1  758.03   131.5  760.46   140.9  761.49   150.3  761.99   159.6  762.35
     169  762.55   178.4  763.56   187.8  766.38   197.2  770.43
#Mann= 3 , 0 , 0
       0      .1       0   100.9    .045       0   115.9     .06       0
Bank Sta=100.9,115.9
XS Rating Curve= 0 ,0
Exp/Cntr=0.3,0.1

Type RM Length L Ch R = 1 ,9240.2  ,21.3,25.5,29.8
XS GIS Cut Line= 3
     1830155.281       479099.87     1830248.181      479153.482
     1830355.815      479189.087
#Sta/Elev= 26
       0   781.9     9.8  776.31    19.5  769.97    29.2  763.45      39  759.05
    48.8  757.91    58.5     758    68.3     758      78  758.09    87.8  758.05
    97.5  757.94   107.3   757.7   116.7  757.43   122.2  756.64   126.2  756.07
   135.6  755.42   137.2  755.66     145  756.82   154.5  759.13   163.9  760.58
   173.4  761.51   182.8  762.06   192.3  762.52   201.7  763.92   211.2  766.65
   220.6  770.14
#Mann= 3 , 0 , 0
       0      .1       0   122.2    .045       0     145     .06       0
Bank Sta=122.2,145
XS Rating Curve= 0 ,0
Exp/Cntr=0.3,0.1

Type RM Length L Ch R = 1 ,9214.7  ,35.1,34.3,34.1
XS GIS Cut Line= 3
     1830134.409      479111.329     1830167.545       479132.31
     1830356.838      479237.818
#Sta/Elev= 30
       0     788     9.8  782.01    19.6  775.83    29.4   769.5    39.2   762.6
    48.6   758.5    58.1  757.78    67.5  758.03    76.9  758.29    86.3  758.42
    95.8  758.49   105.2  758.44   114.6  758.54     124  758.07   133.4  757.27
   137.8  756.85   142.9  756.36   152.3  754.96   152.8  755.05   161.7  756.61
   171.1  759.38   180.6  760.92     190  761.51   199.4  761.82   208.8  761.84
   218.2  762.03   227.7  764.46   237.1  768.51   246.5  773.11   255.9  777.99
#Mann= 3 , 0 , 0
       0      .1       0   142.9    .045       0   161.7     .06       0
Bank Sta=142.9,161.7
XS Rating Curve= 0 ,0
Exp/Cntr=0.3,0.1

Type RM Length L Ch R = 1 ,9180.4  ,121,130.4,138.4
XS GIS Cut Line= 3
     1830107.399      479134.657     1830146.663      479159.663
     1830329.712       479261.69
#Sta/Elev= 30
       0   793.7     9.3  788.77    18.6  783.29    27.9  777.66    37.2  772.11
    46.6  766.22    56.1  760.41    65.6  757.54    75.1  757.12    84.6  757.44
    94.2  757.77   103.7  757.91   113.2  757.81   122.8  757.36   132.3  756.45
   141.8   755.1   148.4  754.57   151.3  754.33   160.9  755.03   163.4   755.2
   170.4  755.69   179.9   757.8   189.4  759.19     199  760.03   208.5  760.93
     218  761.48   227.5  761.35   237.1  762.26   246.6   765.9   256.1  770.72
#Mann= 3 , 0 , 0
       0     .08       0   141.8    .045       0   163.4     .06       0
Bank Sta=141.8,163.4
XS Rating Curve= 0 ,0
Exp/Cntr=0.3,0.1

Type RM Length L Ch R = 1 ,9049.9  ,153.6,138.3,123
XS GIS Cut Line= 3
     1830062.592      479192.017      1830146.36      479290.541
     1830279.606      479360.854
#Sta/Elev= 24
       0   790.2     9.2  786.55    18.5  782.67    27.7  778.26      37  773.15
    46.2  768.89    55.4  765.01    73.9  755.53    83.1  752.69    92.4  751.99
   101.6  753.18   110.8  754.51   120.1  755.37   129.3  755.68   148.2   756.1
     167  756.82   185.8   757.7   214.1  759.52   232.9  760.52   242.3  761.58
   251.7  763.31   261.2   763.7   270.6  765.08     280  767.18
#Mann= 3 , 0 , 0
       0      .1       0    83.1    .045       0   101.6     .07       0
Bank Sta=83.1,101.6
XS Rating Curve= 0 ,0
Exp/Cntr=0.3,0.1

Type RM Length L Ch R = 1 ,8911.7  ,172.1,182.8,193.5
XS GIS Cut Line= 4
     1829926.539      479310.547     1829994.312      479347.641
     1830072.676      479363.224      1830284.07      479452.372
#Sta/Elev= 30
       0  833.48      29  814.88    38.6   808.5    48.3  801.63    57.9  794.38
    67.6  785.68    77.3  774.89    86.1  764.06      95  755.29    99.4  753.12
   103.9   750.9   112.8  750.56   114.4  750.85   130.5  753.65   139.4  754.53
   148.3  754.97   166.7  755.34   195.4  755.33   243.2  755.92   271.9  756.79
   281.4   757.3     291  758.27   300.6   759.7   310.1  760.72   329.2  762.18
   338.8  764.12   348.3  768.29   357.9  772.95   367.5   774.6   386.6   787.6
#Mann= 3 , 0 , 0
       0      .1       0    99.4    .045       0   114.4      .1       0
Bank Sta=99.4,114.4
XS Rating Curve= 0 ,0
Exp/Cntr=0.3,0.1

Type RM Length L Ch R = 1 ,8728.9  ,287.9,281.9,275.3
XS GIS Cut Line= 3
     1829874.923      479454.541     1830014.762      479562.834
     1830157.898      479695.141
#Sta/Elev= 30
       0  826.14    19.6  812.93    29.5  805.45    39.3  797.08    68.8  770.91
    78.6  761.71    88.4  753.16    98.3  747.96   108.1     747   117.9  748.69
   127.7  750.11   137.6  750.87   147.4  751.33   157.2  751.63     167   751.7
   176.9  751.58   196.4   751.6   235.3  752.48   245.1  752.78   254.8  753.39
   264.6  754.22   274.3  755.59   284.1  757.38   293.8  759.52   303.6  761.22
   313.3  762.25   342.6   764.6   352.3  765.98     362  768.77   371.8  772.36
#Mann= 3 , 0 , 0
       0      .1       0    98.3    .045       0   117.9     .08       0
Bank Sta=98.3,117.9
XS Rating Curve= 0 ,0
Exp/Cntr=0.3,0.1

Type RM Length L Ch R = 1 ,8446.9  ,182.6,191.7,200.8
XS GIS Cut Line= 3
     1829716.387      479715.777      1829951.63      479810.395
     1830057.533      479931.923
#Sta/Elev= 30
       0  790.06     9.8  785.81    19.5  780.74    29.3  775.26      39  769.35
    58.5  754.93    68.3  751.22      78  749.72    87.8  747.88    97.5  744.88
   107.3  742.65     117  743.14   126.8  745.65   136.5  747.67     156  747.49
   175.5  747.85   204.8  748.17   253.6  749.75   272.5  750.12     282  750.64
   291.5  752.34     301  754.66   310.4  757.91   329.4  766.52   338.9  771.17
   348.4  776.39   386.3  798.48   395.8  803.82   405.3  808.12   414.8  811.77
#Mann= 3 , 0 , 0
       0      .1       0    97.5    .045       0     117      .1       0
Bank Sta=97.5,117
XS Rating Curve= 0 ,0
Exp/Cntr=0.3,0.1

Type RM Length L Ch R = 1 ,8255.2  ,165,175.5,186
XS GIS Cut Line= 2
     1829592.568      479793.692     1829881.326      480078.744
#Sta/Elev= 30
       0  795.45     9.7  792.16    19.3  788.32    48.3  776.24    67.6  768.75
    77.3  765.18    96.6  758.53   115.9  748.91   135.2  744.12   144.9  741.13
   154.6  739.89   164.2   741.1   173.9  742.94   183.6  743.63   193.2   743.7
   202.9     744   212.5  744.15   222.2  744.01   241.5  744.05   299.5   743.5
   309.2  743.83   318.8  746.78   328.5  752.01   338.1  758.34   347.8  765.63
   367.1  785.26   376.8  793.43   386.4  800.96   396.1  807.82   405.8  812.87
#Mann= 3 , 0 , 0
       0      .1       0   144.9    .045       0   164.2      .1       0
#XS Ineff= 2 , 0
                          209.96          751.81
Permanent Ineff=
       F       F
Bank Sta=144.9,164.2
XS Rating Curve= 0 ,0
Exp/Cntr=0.3,0.1

Type RM Length L Ch R = 1 ,8079.7  ,173.9,166,158.1
XS GIS Cut Line= 4
     1829487.933      479865.934     1829549.817      479960.834
      1829584.77       480063.57     1829704.056      480203.544
#Sta/Elev= 30
       0  813.92    18.9  803.35    28.3   797.6    56.6  780.88    66.1  775.13
    75.5  769.74      85   765.3   113.3  753.46   122.3   749.4   131.4  745.12
   140.4  740.69   149.5  737.75   155.6  737.06   158.5  736.73   167.6  736.95
   170.6  737.43   176.6   738.4   185.6  740.38   194.7  740.86   241.2  741.38
   279.9   741.3   308.9  741.46   318.6  741.64   328.3  742.13     338  742.88
   347.6  745.36   376.7  762.61   386.4  769.85     396  777.87   405.7  785.39
#Mann= 3 , 0 , 0
       0      .1       0   155.6    .045       0   170.6      .1       0
Bank Sta=155.6,170.6
XS Rating Curve= 0 ,0
Exp/Cntr=0.3,0.1

Type RM Length L Ch R = 1 ,7913.7  ,275.3,274.7,273.8
XS GIS Cut Line= 3
     1829325.326      479946.862     1829448.937      480103.112
     1829554.768      480290.434
#Sta/Elev= 30
       0  798.78     9.5  793.02    28.5  781.12      38  774.98    56.9  762.57
    66.4  756.52    75.9  750.87    85.4  745.48    94.9  740.86   104.4   738.5
   113.8  738.23   123.3  736.77   132.8  734.75   142.3  734.06   150.1  735.26
   151.8  735.52   161.3  737.76   170.8  739.07   180.3  739.44   199.2  739.67
   238.4  739.32   277.5  739.79   287.2  740.15     297  740.71   306.8  741.09
   316.6  741.19   326.4  741.52   345.9  742.44   394.8  745.44   414.4  746.85
#Mann= 3 , 0 , 0
       0      .1       0   132.8    .045       0   150.1      .1       0
#XS Ineff= 2 , 0
                           199.6          740.87
Permanent Ineff=
       F       F
Bank Sta=132.8,150.1
XS Rating Curve= 0 ,0
Exp/Cntr=0.3,0.1

Type RM Length L Ch R = 1 ,7639    ,261.4,261.6,261.8
XS GIS Cut Line= 2
     1829104.332      480073.642     1829405.878      480430.358
#Sta/Elev= 30
       0  837.45    29.2  819.53    38.9  813.68    58.4  802.04    87.6  784.95
    97.3  778.65     107  771.06   116.8  762.69   126.5  753.82   136.2  743.14
     146  733.95   151.3  732.17   155.7  730.69   165.4  730.95   166.3   731.1
   175.2   732.6   184.9  733.92   194.6  734.72   214.1   735.8     253  736.08
   291.9  736.53   350.3  737.41     360  737.58   379.5  738.37   389.2   738.4
     399  738.61   408.7  739.01   418.4  739.83   457.4  743.81   467.1  744.61
#Mann= 3 , 0 , 0
       0      .1       0   151.3    .045       0   166.3      .1       0
Bank Sta=151.3,166.3
XS Rating Curve= 0 ,0
Exp/Cntr=0.3,0.1

Type RM Length L Ch R = 1 ,7377.4  ,303.3,298.1,292.9
XS GIS Cut Line= 3
      1828948.51      480172.086     1828960.229      480304.898
     1829225.854      480626.513
#Sta/Elev= 30
       0  824.76    28.6  809.76    47.6  799.48    76.2  783.34   104.8  767.53
   133.3  751.15     143  748.02   152.7  741.95   162.4  735.19   172.1  731.18
   181.8  728.91   191.5  727.23   201.2  727.63   206.5  728.79   220.6     732
   230.3  732.41   259.4   732.1   288.5  732.02   327.3  731.66   346.7   731.2
   375.8  730.82   404.9   731.1   424.4  731.47   482.6  733.11   492.2  735.02
     502  738.87   521.4  748.23     531  753.08   540.8  758.77   550.4  765.55
#Mann= 3 , 0 , 0
       0      .1       0   181.8    .045       0   206.5      .1       0
Bank Sta=181.8,206.5
XS Rating Curve= 0 ,0
Exp/Cntr=0.3,0.1

Type RM Length L Ch R = 1 ,7079.4  ,446.2,441,435.5
XS GIS Cut Line= 3
     1828707.625       480502.26     1828906.236      480652.954
     1829051.375      480825.176
#Sta/Elev= 30
       0  803.44    28.8   786.5    38.4  780.63    47.9   774.3    57.5  767.52
    67.1  759.75    86.3  739.49    95.9  730.72   105.5  724.99     113  723.29
   115.1  722.81   124.6  723.39     128  723.81   134.2  724.58   143.8  725.33
   191.8  726.81   249.3  727.36   298.3  726.68   327.6  726.87   337.4  727.15
     357  728.65   376.6  730.61   386.4  732.46   396.2  738.22     406   745.5
   415.8  753.21   425.6  761.45   435.4  770.22   445.2  777.79   474.5  797.36
#Mann= 3 , 0 , 0
       0      .1       0     113    .045       0     128      .1       0
Bank Sta=113,128
XS Rating Curve= 0 ,0
Exp/Cntr=0.3,0.1

Type RM Length L Ch R = 1 ,6638.4  ,353.3,365.2,377
XS GIS Cut Line= 2
     1828594.458      480940.462     1829012.512      481125.173
#Sta/Elev= 30
       0  771.71     9.7  766.07    19.4  760.05    29.2  754.17    38.9  748.17
    48.6  742.29    68.1  731.41    77.8  726.35    87.5  722.64    97.2  720.58
     107  718.82   116.7  717.85   126.4  718.42   136.1  718.96   155.6   719.7
   213.9   722.3   233.4  723.05   243.1  724.91   252.8  728.78   291.7  747.42
   301.4  752.25   311.2  757.98   320.9  764.41   350.1  784.31   359.8  790.75
   369.5  797.01   379.2  803.11   398.7  814.99   427.9  832.24     457  849.65
#Mann= 3 , 0 , 0
       0      .1       0     107    .045       0   126.4     .07       0
Bank Sta=107,126.4
XS Rating Curve= 0 ,0
Exp/Cntr=0.3,0.1

Type RM Length L Ch R = 1 ,6273.2  ,238.4,240.8,242.8
XS GIS Cut Line= 3
      1828381.39      481181.038     1828458.473      481237.982
     1828629.306      481471.315
#Sta/Elev= 25
       0  812.44     9.6  805.54    28.8  791.96    47.9  778.26    67.1  764.41
    76.7  757.33    86.2     750    95.8  742.19   105.5  733.91   115.1  724.18
   124.8  715.52   129.5  713.66   134.4  711.73     144  711.65   144.5  711.67
   153.7  712.11     173  713.26   192.2  714.09   221.2     715   250.1  715.62
   288.6   716.2   298.3  716.57   307.9  717.05   336.8  718.82     385  721.26
#Mann= 3 , 0 , 0
       0      .1       0   129.5    .045       0   144.5      .1       0
Bank Sta=129.5,144.5
XS Rating Curve= 0 ,0
Exp/Cntr=0.3,0.1

Type RM Length L Ch R = 1 ,6032.4  ,384.7,390.7,396.7
XS GIS Cut Line= 3
     1828236.164      481325.699      1828327.31      481479.779
     1828366.372       481657.73
#Sta/Elev= 27
       0  778.11     9.4  772.62    18.8  766.64    28.3   758.8    37.7  748.72
    47.1  739.22    56.5  730.01      66  719.54    75.4  710.73    84.8  706.89
    94.2  706.94   101.2  707.14   131.9  708.03   141.3  708.53   160.2   711.9
   169.6   712.6     179  712.55   188.6  711.91   198.2  711.56   207.8  711.86
   217.4  712.34   284.5  714.66   322.8  716.13   332.4  716.94     342  718.14
   351.6  719.39   361.2  721.05
#Mann= 3 , 0 , 0
       0      .1       0    84.8    .045       0   101.2      .1       0
Bank Sta=84.8,101.2
XS Rating Curve= 0 ,0
Exp/Cntr=0.3,0.1

Type RM Length L Ch R = 1 ,5641.7  ,338.6,344.1,349.7
XS GIS Cut Line= 3
      1827900.14      481467.149      1827968.89      481717.843
     1827975.834      481830.343
#Sta/Elev= 29
       0  748.46     9.6  742.71    19.3  736.17    28.9  729.35    38.5  722.75
    48.1  716.44    57.8   710.2    67.4  705.38      77   703.6    86.6   703.4
    97.1  703.47   115.5  703.81   125.2  704.22   134.8  705.41   144.4  706.46
     154  706.95   173.3   708.2   192.6  709.06   221.4  710.96     260   713.9
   269.3   714.8   278.7  716.21   288.1  718.08   306.9  722.14   316.3   724.3
   325.7  727.27   335.1   731.3   363.3  745.67   372.7  750.33
#Mann= 3 , 0 , 0
       0      .1       0      77    .045       0    97.1     .07       0
Bank Sta=77,97.1
XS Rating Curve= 0 ,0
Exp/Cntr=0.3,0.1

Type RM Length L Ch R = 1 ,5297.6  ,287,287.4,287.7
XS GIS Cut Line= 3
     1827583.876      481481.052     1827588.386      481689.355
     1827574.445      481833.121
#Sta/Elev= 30
       0  761.41     9.5  758.93    18.9  756.06    28.4  752.38    37.9  747.97
    47.4  742.94    75.8  726.18   104.2  709.09   113.6  702.94   123.1  699.66
   132.6  699.19   142.1  699.47   151.5   699.5     161  699.15   170.5  699.99
   179.9     703   198.9  711.34   208.4  714.66     218  717.18   237.2  721.62
   256.5  725.58   266.1  727.81   275.8  730.32   285.4  732.95     295  735.83
   304.6  739.39   314.3  743.53   323.9  747.25   343.2  753.77   352.8  757.32
#Mann= 3 , 0 , 0
       0      .1       0   123.1    .045       0   142.1      .1       0
Bank Sta=123.1,142.1
XS Rating Curve= 0 ,0
Exp/Cntr=0.3,0.1

Type RM Length L Ch R = 1 ,5010.2  ,210,206.6,203.1
XS GIS Cut Line= 3
     1827335.556      481447.704     1827301.529      481580.343
     1827302.917      481826.177
#Sta/Elev= 30
       0  749.19     9.8  744.47    19.6  738.42    39.1  724.28    48.9  717.88
    68.5   706.2    78.2  700.88      88  697.93    97.8  697.16   146.8  695.96
   170.8  695.07   176.3  694.85   186.1  694.68   195.9  694.69   215.6  695.61
   235.3  695.71   245.1  696.31   254.9   696.4   264.8  695.97   274.6  695.87
   284.4   696.8   294.3  698.82   304.1  701.39   313.9  704.43   323.8  708.17
   333.6  712.84   343.4  718.27   353.3  724.14   372.9  736.29   382.8  742.33
#Mann= 3 , 0 , 0
       0      .1       0   170.8    .045       0   195.9      .1       0
Bank Sta=170.8,195.9
XS Rating Curve= 0 ,0
Exp/Cntr=0.3,0.1

Type RM Length L Ch R = 1 ,4803.6  ,158,159.1,160.1
XS GIS Cut Line= 3
     1827134.167       481403.26     1827086.945      481576.871
     1827120.279       481784.51
#Sta/Elev= 30
       0  731.36     9.5  728.99    18.9  725.35    28.4  720.66    47.4   710.5
    56.8   706.1    66.3  703.86    75.8   703.1    85.2  701.55    94.7  700.77
   113.6  700.57     142  699.36     161  698.41   208.6  695.27   218.2  694.22
   227.7  692.48   236.6  691.12   237.3  691.01   251.6  691.44   256.4  691.68
     266   693.4   275.5  694.88   285.1  695.47   313.7  695.56   332.9  694.56
   342.4  695.12     352  697.67   361.5  702.41   371.1  709.25   390.2  725.16
#Mann= 3 , 0 , 0
       0      .1       0   236.6    .045       0   251.6      .1       0
Bank Sta=236.6,251.6
XS Rating Curve= 0 ,0
Exp/Cntr=0.3,0.1

Type RM Length L Ch R = 1 ,4644.6  ,140.2,111.3,81
XS GIS Cut Line= 3
     1826875.834      481330.343     1826930.001      481535.899
     1826960.556      481801.177
#Sta/Elev= 30
       0  734.36      29  723.39    48.3  716.41      58  713.18    67.6   710.8
    77.3  709.18      87  708.13   125.6   704.8   135.3  704.18   164.3  703.31
   183.6  702.42   212.6  700.44   241.2  698.18   288.9  695.13   298.4  693.96
   307.9  692.44   317.5   691.3     327  690.55   355.6  688.88   365.2  688.55
   374.8  689.05   393.8  691.94   403.3  692.14   422.4  691.45   431.9  691.34
   441.5  691.62     451  695.27   460.5  703.44   470.1  712.93   479.6   722.7
#Mann= 3 , 0 , 0
       0      .1       0   355.6    .045       0   374.8      .1       0
Bank Sta=355.6,374.8
XS Rating Curve= 0 ,0
Exp/Cntr=0.3,0.1

Type RM Length L Ch R = 1 ,4533.3  ,44.2,39.7,39.8
XS GIS Cut Line= 4
     1826674.445      481523.399     1826805.371      481698.928
     1826889.506      481719.638     1826937.361      481801.623
#Sta/Elev= 30
       0  708.38     9.5  704.29      19  700.81    28.6  698.03    38.1   695.6
    47.6  693.96    57.1  693.13    76.2  692.07    85.7  691.81   133.3  691.42
   152.3   691.1   161.8   690.9   180.9  689.96   190.4  689.64   199.9  689.68
   209.5  690.03     219  690.11   228.6  689.92   238.2  689.18   247.9  688.25
   257.5  688.18   267.1  689.49   276.7  690.24   286.4  690.42   315.1  690.44
   343.6  690.09   362.6  690.07   372.1  692.81   381.6  699.45   400.6  717.55
#Mann= 3 , 0 , 0
       0     .08       0   238.2    .045       0   267.1      .1       0
Bank Sta=238.2,267.1
XS Rating Curve= 0 ,0
Exp/Cntr=0.3,0.1

Type RM Length L Ch R = 1 ,4493.6  ,220.5,245.3,266.3
XS GIS Cut Line= 4
     1826634.862       481540.76     1826778.818      481732.285
     1826869.103      481754.509     1826910.652      481824.623
#Sta/Elev= 30
       0  707.88     9.6  702.26    19.2  698.32    28.8  695.92    47.9  692.73
    57.5   691.5    67.1  690.73    95.8  689.35     115  688.91   143.8   687.9
   172.5  687.77   191.7  687.06   201.3  687.18   210.8  687.69     230  689.15
   239.6  689.22   267.5  688.41   291.2  687.47   295.4  687.32   304.7  687.42
   306.2  687.63     314  688.71   323.3  689.21   359.7  689.58   368.8  690.84
   377.8  695.45   386.9  703.81     396  712.84     405  722.02   414.1  730.89
#Mann= 3 , 0 , 0
       0     .08       0   291.2    .045       0   306.2      .1       0
Bank Sta=291.2,306.2
XS Rating Curve= 0 ,0
Exp/Cntr=0.3,0.1

Type RM Length L Ch R = 1 ,4248.3  ,342,345.6,349
XS GIS Cut Line= 2
     1826523.918      481647.771     1826663.345      481930.667
#Sta/Elev= 30
       0  704.57     9.6  700.01    19.1  696.58    28.7  694.75    38.2  693.25
    57.3  689.66    66.9  688.03    76.5  686.91      86   686.2   105.1   685.4
   114.7   685.4   124.2  685.18   143.4  683.78   162.5   683.4     172  682.81
   181.6  681.88   187.6  681.45   191.1   681.2   200.7   681.2   202.6  681.46
   210.3   682.5   219.8   684.1   229.4  684.53   238.9  684.14   248.5  684.37
     258  686.28   267.6  689.18   277.2  693.95   296.3   705.4   315.4  716.05
#Mann= 3 , 0 , 0
       0      .1       0   187.6    .045       0   202.6      .1       0
Bank Sta=187.6,202.6
XS Rating Curve= 0 ,0
Exp/Cntr=0.3,0.1

Type RM Length L Ch R = 1 ,3902.7  ,193.6,194.7,195.7
XS GIS Cut Line= 2
      1826226.21      481721.315     1826356.765      482130.343
#Sta/Elev= 30
       0  747.26     9.8  741.59    19.5  735.35    29.3  728.36      39  721.23
    48.8   714.7    58.6     709    68.3  703.84    78.1     699    87.8  694.52
   107.3  685.82   117.1  681.91   126.9   679.9   133.7  679.47   136.6  679.28
   148.7  679.65   185.4  680.02   214.7  679.98     244  680.16   253.7  680.52
   273.2  683.04   302.5  683.85   341.5   682.7   351.3  683.46     361  685.98
   380.6  694.34   390.3  698.26   409.8  706.49   419.6  711.32   429.4  717.32
#Mann= 3 , 0 , 0
       0      .1       0   133.7    .045       0   148.7      .1       0
Bank Sta=133.7,148.7
XS Rating Curve= 0 ,0
Exp/Cntr=0.3,0.1

Type RM Length L Ch R = 1 ,3708.1  ,331.7,331,330.1
XS GIS Cut Line= 2
     1826053.293      481794.232     1826148.432      482147.704
#Sta/Elev= 30
       0  752.25    19.3  740.08    28.9  733.37    38.5  725.86    48.2  718.41
    57.8  711.17    67.4  704.27    77.1  697.78    86.7  691.81    96.3  686.51
     106   681.9   115.6   677.8   125.2  674.79   134.9   673.7   144.5  673.46
   154.1  673.91   173.4  677.32     183  678.12   221.6  678.91   231.2  678.99
   240.8  679.85   250.5  682.88   260.1   684.9   269.7   685.6     289  686.56
   308.2  687.46   327.5  688.12   337.2  688.68   346.8  689.37     366  691.23
#Mann= 3 , 0 , 0
       0      .1       0   134.9    .045       0   154.1      .1       0
Bank Sta=134.9,154.1
XS Rating Curve= 0 ,0
Exp/Cntr=0.3,0.1

Type RM Length L Ch R = 1 ,3377.1  ,283.3,279.9,276.5
XS GIS Cut Line= 2
     1825739.231      481901.003     1825826.036      482183.121
#Sta/Elev= 26
       0  719.92    19.7  704.59    29.5  696.41    49.2  679.42      59  673.66
    68.9  671.76    88.6  669.27    98.4  669.03   105.7  670.18   108.2  670.57
   118.1  672.56   127.9  673.29   147.6  673.48   167.3  673.51   177.1   673.6
   186.9  673.87   196.8  674.32   206.6  674.65   226.3  674.41   236.1  676.67
     246  680.63   255.8  684.68   265.6  688.08   275.5   689.8   285.3  690.62
   295.2   691.3
#Mann= 3 , 0 , 0
       0      .1       0    88.6    .045       0   105.7      .1       0
#XS Ineff= 2 , 0
                          206.73             677
Permanent Ineff=
       F       F
Bank Sta=88.6,105.7
XS Rating Curve= 0 ,0
Exp/Cntr=0.3,0.1

Type RM Length L Ch R = 1 ,3097.2  ,175.7,145.6,96.7
XS GIS Cut Line= 2
     1825449.155      481976.784     1825574.051      482235.228
#Sta/Elev= 26
       0  685.91     9.6     679    19.1  674.54    28.7  671.74    38.3  669.96
    47.8  669.27      67   668.9    86.1  668.22    95.7  668.25   114.8  668.83
   124.4  668.52   143.5   664.6   153.1  664.25   162.7  664.53   172.2  665.03
   181.8  666.36   191.4  667.99   200.9  668.75   210.5  668.84   220.1  668.44
   229.6  668.88   239.2  672.18   258.3  680.13   267.9  683.97   277.5  686.97
     287  688.33
#Mann= 3 , 0 , 0
       0      .1       0   143.5    .045       0   162.7      .1       0
#XS Ineff= 2 , 0
          114.63  669.76
Permanent Ineff=
       F       F
Bank Sta=143.5,162.7
XS Rating Curve= 0 ,0
Exp/Cntr=0.3,0.1

Type RM Length L Ch R = 1 ,2951.6  ,105.5,62.2,81.5
XS GIS Cut Line= 4
     1825186.918      482040.138      1825275.46      482175.555
     1825511.187       482151.71       1825553.8      482246.607
#Sta/Elev= 30
       0  681.47     9.5   680.6      19  678.78    28.6  675.92    38.1   672.5
    47.6  669.45    57.1  667.68   114.2  664.99   133.2  664.46   152.3  664.64
   209.2  666.16   228.1  666.51   237.6  666.23   247.1   664.9   256.6  663.07
     266  662.64   277.5  663.45   322.9  666.24   332.4  666.62   370.3   666.8
   398.7  667.32   408.2  668.44   417.6  668.68   427.1  668.38   436.6  668.55
     446  670.96   474.4  682.34   483.8  685.59   493.3   687.5   502.8  688.18
#Mann= 3 , 0 , 0
       0      .1       0   256.6    .045       0   277.5      .1       0
Bank Sta=256.6,277.5
XS Rating Curve= 0 ,0
Exp/Cntr=0.3,0.1

Type RM Length L Ch R = 1 ,2889.4  ,125.4,209.1,248
XS GIS Cut Line= 4
     1825171.293      482085.277     1825278.064       482226.77
     1825508.099      482203.332     1825536.745      482294.478
#Sta/Elev= 30
       0  668.97     9.3  667.49    18.7  666.71    65.3  664.88    93.3  663.21
   102.6  662.91     112  662.99   130.6  664.35   139.9  664.65   149.3  664.62
   158.6  664.03   177.3   660.3   215.8  661.04   225.4  660.97   245.5   661.2
   260.5  661.63   273.6  662.04   283.2  662.78   292.9  663.96   312.1  665.92
   321.8  666.85   331.4  667.56   360.3  669.01   398.8  671.62   408.5  672.18
   437.2   683.2   446.7  686.06   456.2  687.46   465.8  687.89     504  689.01
#Mann= 3 , 0 , 0
       0      .1       0   245.5    .045       0   260.5      .1       0
Bank Sta=245.5,260.5
XS Rating Curve= 0 ,0
Exp/Cntr=0.3,0.1

Type RM Length L Ch R = 1 ,2680.3  ,321.1,317.8,314.2
XS GIS Cut Line= 2
     1825149.634      482088.795     1825156.925      482358.587
#Sta/Elev= 26
       0  668.38     9.6  666.78    19.3  665.98    28.9  665.32    48.2  664.16
    86.8  662.04    96.4  661.96     106  662.17   115.7  662.71   125.3  662.86
     135  662.42   144.6  661.56   154.2  659.27   163.9  657.78   168.4  657.33
   173.5  656.82   183.4  657.27   192.8  659.14   202.4  663.41   212.1  668.16
   221.7  673.18   231.3  678.56     241  682.96   250.6  685.02   260.2  685.47
   269.9  685.57
#Mann= 3 , 0 , 0
       0      .1       0   168.4    .045       0   183.4      .1       0
Bank Sta=168.4,183.4
XS Rating Curve= 0 ,0
Exp/Cntr=0.3,0.1

Type RM Length L Ch R = 1 ,2362.5  ,380.8,379.4,377.7
XS GIS Cut Line= 2
      1824815.62      482159.683     1824857.663      482390.726
#Sta/Elev= 27
       0  662.62     9.8   662.4    19.6  662.12    29.4  661.92    39.1  661.69
    48.9   661.2    58.7  660.16    68.5  658.85    78.3  658.37    88.1  658.61
    97.8  658.12   107.6  655.06   117.4  650.94     120  650.62   127.2  649.75
     135  650.57     137  650.78   146.8  653.57   156.6  656.82   166.3  661.44
   176.1  667.28   185.9  673.25   195.7  677.71   205.5   679.1   215.3  679.42
     225  679.59   234.8  679.82
#Mann= 3 , 0 , 0
       0      .1       0     120    .045       0     135      .1       0
Bank Sta=120,135
XS Rating Curve= 0 ,0
Exp/Cntr=0.3,0.1

Type RM Length L Ch R = 1 ,1983.1  ,231.1,234.2,237.3
XS GIS Cut Line= 2
     1824440.302      482246.976     1824503.496      482499.754
#Sta/Elev= 30
       0  655.06     9.6  654.96    19.3  654.69      29  653.92    38.6  653.13
    48.2  653.46    57.9  654.08    67.6  653.96    77.2  653.36    86.8  652.68
    96.5  651.98   106.2  651.27   115.8  650.58   125.4  649.01   135.1  646.47
   144.8  645.02   144.9  645.03   154.4  645.61   159.9  646.86     164   647.8
   173.7  651.13   183.4  654.86     193  659.32   202.7  664.71   212.3  670.76
     222  676.42   231.6  680.52   241.3  683.53   250.9  686.18   260.6  687.26
#Mann= 3 , 0 , 0
       0      .1       0   135.1    .045       0   154.4      .1       0
Bank Sta=135.1,154.4
XS Rating Curve= 0 ,0
Exp/Cntr=0.3,0.1

Type RM Length L Ch R = 1 ,1748.8  ,91.8,92.1,92.4
XS GIS Cut Line= 3
      1824268.19      482237.504     1824237.547      482352.612
     1824254.696      482510.391
#Sta/Elev= 30
       0  657.79     9.2  654.63    18.3  652.65    27.5  652.39    36.6  652.32
    45.8  651.56      55  650.29    64.1  649.51    73.3  649.46    82.5  649.58
    91.6  649.49     110  649.03   119.1  648.72   128.4  647.87   137.8  646.62
   147.1  645.98   165.8  645.55   175.1  644.44   184.5  643.03   186.4  642.84
   193.8  642.12   203.1  642.83   212.5  645.37   221.8  647.62   231.2  648.48
   240.5  649.07   249.8  649.81   259.2  651.48   268.5  655.25   277.8  660.46
#Mann= 3 , 0 , 0
       0     .06       0   186.4    .045       0   203.1      .1       0
Bank Sta=186.4,203.1
XS Rating Curve= 0 ,0
Exp/Cntr=0.3,0.1

Type RM Length L Ch R = 1 ,1656.7  ,26,26,26
XS GIS Cut Line= 3
     1824137.936      482257.066     1824143.711      482324.566
     1824162.895      482530.467
#Sta/Elev= 24
       0     651    19.4  649.46    38.7  647.05    48.4  646.91    58.1  647.34
    67.8  647.06    77.2  646.44    86.6  646.03   105.4  645.84   133.5  645.36
   152.3  645.32   161.7  644.38   171.1  642.53   175.7  641.78   180.5     641
   189.9  641.44   190.7  641.67   199.3  644.09   208.7  646.61   218.1  647.61
   246.3  649.06   255.7  649.95   265.1  652.25   274.5  656.15
#Mann= 3 , 0 , 0
       0      .1       0   175.7    .045       0   190.7      .1       0
Bank Sta=175.7,190.7
XS Rating Curve= 0 ,0
Exp/Cntr=0.3,0.1

Type RM Length L Ch R = 1 ,1630.8  ,104.2,101.6,98.8
XS GIS Cut Line= 3
     1824110.693      482256.447     1824118.093      482329.116
     1824136.853      482530.467
#Sta/Elev= 24
       0  650.87    18.3  649.47    27.4   648.5    36.5  646.85    45.6  646.12
    54.8  646.57    63.9  646.68    82.7  646.19   101.9  645.85   130.8   645.1
   150.1  644.72   159.7  644.21   169.3  642.64   178.1  640.89     179  640.71
   188.6  640.52   193.1  641.48   198.2  642.57   207.9  645.64   217.5  647.28
   236.8  648.23     256  649.47   265.6  650.56   275.3  653.46
#Mann= 3 , 0 , 0
       0      .1       0   178.1    .045       0   193.1      .1       0
#XS Ineff= 2 , 0
           63.95   647.3
Permanent Ineff=
       F       F
Bank Sta=178.1,193.1
XS Rating Curve= 0 ,0
Exp/Cntr=0.3,0.1

Type RM Length L Ch R = 1 ,1529.2  ,172,171.6,171.2
XS GIS Cut Line= 3
     1823986.635      482218.626     1823993.182       482290.27
     1824047.009      482542.186
#Sta/Elev= 24
       0  665.85      18  657.32      27  653.26      36  650.61      45  649.66
      63  648.19    71.9  646.53    81.5  645.12      91  645.04   100.6  645.29
   110.1  645.27   157.8  644.61   205.5  643.66     215  643.34   224.6  642.06
   234.1  640.58   243.7  639.75   253.2  640.85   262.8  644.03   272.3  646.16
   281.8  646.78   310.5  647.43     320  647.72   329.5  648.13
#Mann= 3 , 0 , 0
       0     .06       0   234.1    .045       0   253.2      .1       0
#XS Ineff= 2 , 0
          103.36  647.25
Permanent Ineff=
       F       F
Bank Sta=234.1,253.2
XS Rating Curve= 0 ,0
Exp/Cntr=0.3,0.1

Type RM Length L Ch R = 1 ,1357.6  ,66.1,63.9,61.6
XS GIS Cut Line= 3
     1823837.569      482225.421     1823816.963      482302.766
     1823908.448      482697.718
#Sta/Elev= 30
       0  657.11     8.9  651.46    17.8  647.35    26.7  645.66    35.6  645.18
    62.3   644.6    99.4  643.45   157.3  642.66   195.9  642.75   215.2  643.05
   224.8  642.92   234.5  642.52   244.1   641.8   253.8  640.53   263.4  638.35
   273.1  637.12   282.8  636.99   292.4  637.78     302  641.21   311.7  642.96
   321.4  643.68     331  644.09   369.6  644.88   388.9  644.94   417.9  644.48
   437.2  644.72   446.8  646.36   456.5  650.28   475.8  660.02   485.4  665.41
#Mann= 3 , 0 , 0
       0     .07       0   263.4    .045       0   292.4      .1       0
#XS Ineff= 2 , 0
          215.65  646.78
Permanent Ineff=
       F       F
Bank Sta=263.4,292.4
XS Rating Curve= 0 ,0
Exp/Cntr=0.3,0.1

Type RM Length L Ch R = 1 ,1293.6  ,49,49.1,48.9
XS GIS Cut Line= 3
     1823754.754      482191.446     1823729.781      482305.522
      1823862.54      482697.375
#Sta/Elev= 30
       0  663.19    19.5  650.46    29.2  645.65    38.9  643.62    48.7  643.21
    97.3  642.53   126.4  642.41   145.6  642.49   193.8   642.4   232.2  643.05
   241.9  643.08   270.7  642.72   280.4  642.85     290  643.57   299.6  643.87
   309.2  642.52   318.8  638.93   328.4  637.18   338.1  636.98   347.7  637.97
   366.9   642.3   386.2   643.4   395.8   643.7   424.7  643.71   443.9  644.03
     492  643.74   501.6     644   511.3  645.55   520.9   649.5   530.5  654.64
#Mann= 3 , 0 , 0
       0     .08       0   318.8    .045       0   347.7      .1       0
#XS Ineff= 2 , 0
          299.15  646.15
Permanent Ineff=
       F       F
Bank Sta=318.8,347.7
XS Rating Curve= 0 ,0
Exp/Cntr=0.3,0.1

Type RM Length L Ch R = 1 ,1244.6  ,69.1,76.2,83.3
XS GIS Cut Line= 2
     1823638.389      482189.322     1823815.882      482711.481
#Sta/Elev= 30
       0   653.4    19.4  645.96      29  643.54    38.7  642.39    48.4  641.91
    67.7   641.7   106.4   641.8   125.8  642.09   145.1  641.92   164.5  642.05
   183.8  641.73   203.2   641.7   232.2  641.92   280.6  642.96   299.9  642.95
   319.3  642.64     329  641.97   338.6  639.17   348.3  635.91     358   635.8
   367.7  638.78   377.3   641.2     387  642.05   435.4  642.09   493.4  642.85
   512.8  643.35   522.5  643.34   532.2  644.11   541.8  648.06   551.5  654.46
#Mann= 3 , 0 , 0
       0      .1       0   338.6    .045       0   367.7      .1       0
#XS Ineff= 2 , 0
          290.23     645  396.03           644.5
Permanent Ineff=
       F       F
Bank Sta=338.6,367.7
XS Rating Curve= 0 ,0
Exp/Cntr=0.3,0.1
